--- LitLaurCk.prj (project) ---

Proj Title=LitLaurCk
Current Plan=p01
Default Exp/Contr=0,0
English Units
Geom File=g01
Flow File=f01
Plan File=p01
BEGIN DESCRIPTION:
END DESCRIPTION:
DSS Export Rating Curves= 0
DSS Export Rating Curve Sorted= 0
DSS Export Volume Flow Curves= 0
DXF OffsetX= 0
DXF OffsetY= 0
DXF ScaleX= 0
DXF ScaleY= 0

--- LitLaurCk.p01 (plan) ---

Plan Title=Floodplain
Program Version=4.00
Geom File=g01
Flow File=f01
K Sum by GR=0
Std Step Tol=0.01
Critical Tol=0.01
Num of Std Step Trials=20
Max Error Tol=0.3
Flow Tol Ratio=0.001
Split Flow NTrial=30
Split Flow Tol=0.02
Split Flow Ratio=0.02
Log Output Level=0
Friction Slope Method=1
Unsteady Friction Slope Method=2
Unsteady Bridges Friction Slope Method=1
Global Log Level=0
CheckData=False
Run HTab=0
Run UNet=0
Run PostProcess=0
UNET Theta=0
UNET Theta Warmup=0
UNET ZTol=0
UNET ZSATol=0
UNET MxIter=0
UNET MaxInSteps=0
UNET DtIC=0
UNET DtMin=0
UNET MaxCRTS=0
UNET WFStab=0
UNET SFStab=0
UNET WFX=0
UNET SFX=0
UNET DSS MLevel=0
UNET DZMax Abort=0
UNET Convert EG Bridges=0
UNET Use Existing IB Tables=0
UNET Froude Limit=0
UNET Froude Power=0
Write IC File=0
Echo Input=False
Echo Output=False
Write Detailed=0

--- LitLaurCk.f01 (steady flow) ---

Flow Title=NFF Regression Equation
Program Version=4.00
Number of Profiles=1
Profile Names=P100yr
River Rch & RM=LitLaurCk,Main      ,31992.5
578.2807
River Rch & RM=LitLaurCk,Main      ,30283.1
608.2601
River Rch & RM=LitLaurCk,Main      ,29602.4
703.7758
River Rch & RM=LitLaurCk,Main      ,27604.4
736.1474
River Rch & RM=LitLaurCk,Main      ,24870.8
816.5054
River Rch & RM=LitLaurCk,Main      ,20649.8
887.7087
River Rch & RM=LitLaurCk,Main      ,20210.8
996.3252
River Rch & RM=LitLaurCk,Main      ,16762.7
1078.020
River Rch & RM=LitLaurCk,Main      ,16481.2
1198.597
River Rch & RM=LitLaurCk,Main      ,11576.9
1265.195
River Rch & RM=LitLaurCk,Main      ,11088.8
1460.042
River Rch & RM=LitLaurCk,Main      ,6570.2
1575.408
River Rch & RM=LitLaurCk,Main      ,6010.9
2091.256
River Rch & RM=LitLaurCk,Main      ,3013.5
2318.702
River Rch & RM=LitLaurCk,Main      ,27.9
2420.492
Boundary for River Rch & Prof#=LitLaurCk,Main      ,1
Up Type=0
Dn Type=3
Dn Slope=0.02672

--- LitLaurCk.g01 (geometry) ---

Geom Title=USGS 10m DEM
Program Version=4.00

River Reach=LitLaurCk       ,Main
Reach XY= 30
     2114726.547      423871.573     2114439.784      425635.318
     2113779.359      426034.199     2113478.578      425842.792
     2113337.953      426112.323     2112317.749      426241.723
     2111564.179      426745.867     2111263.256      427280.201
      2111471.41       429487.61     2111757.699      429761.072
     2111303.136      430071.895     2111370.518      431136.203
     2110397.754      432867.107     2108867.772      434204.044
     2107834.255      433783.145      2107439.72      433851.057
     2106908.573      434573.704     2106632.355      434577.811
     2105569.582      435613.886     2105206.083      435681.658
     2104920.624      435182.616     2103769.342      434447.222
     2101830.882      434041.804     2100585.332      432752.101
     2099987.715       431406.95     2099669.397      431381.279
      2099425.29      431000.932     2097434.042       430463.74
     2096867.023      430910.908      2096164.83       431084.37

Type RM Length L Ch R = 1 ,31992.5 ,299.1,302.8,303.3
XS GIS Cut Line= 3
      2114505.08      423818.576     2114723.795      423881.187
      2114942.51      423943.798
#Sta/Elev= 24
       0 3038.52    49.5 3034.46   138.5 3027.35   197.8 3022.74   207.7 3022.23
   209.33022.225   217.6  3022.2   227.5 3022.58   244.33023.508   257.2 3024.06
   267.1 3024.39   306.6 3025.42   326.4 3026.07   346.2 3027.06   356.1 3027.73
     366 3028.52   385.8 3030.37   395.6 3031.46   405.5 3032.68   415.4 3034.04
   425.3 3035.52   435.2 3037.14   445.1 3038.96     455 3040.91
#Mann= 3 , 0 , 0
       0      .1       0   209.3    .045       0   244.3      .1       0
Bank Sta=209.3,244.3
XS Rating Curve= 0 ,0
Exp/Cntr=0.3,0.1

Type RM Length L Ch R = 1 ,31689.7 ,217.1,211.8,206.5
XS GIS Cut Line= 2
     2114345.308      424079.861      2114901.32      424232.102
#Sta/Elev= 30
       0 3069.76    19.9 3061.94    29.8 3058.28    49.7  3051.5    59.6 3048.39
    79.5 3042.89    89.4 3040.49    99.4 3038.34   109.3 3036.48   139.2 3031.94
   149.1 3030.63     159 3029.92   178.9 3028.82   218.7 3025.82   298.2  3018.4
   337.43015.552   347.9 3015.11   357.8 3015.26   367.8 3016.22   372.43016.829
   417.4 3022.38   437.3 3025.28   457.2  3028.7     487 3034.93     497 3036.72
   506.9 3037.95   516.8 3038.95   526.8 3040.24   556.6 3045.56   576.5 3049.59
#Mann= 3 , 0 , 0
       0      .1       0   337.4    .045       0   372.4      .1       0
Bank Sta=337.4,372.4
XS Rating Curve= 0 ,0
Exp/Cntr=0.3,0.1

Type RM Length L Ch R = 1 ,31477.9 ,335.9,335.7,335.4
XS GIS Cut Line= 2
     2114250.424      424368.148     2114826.464      424390.604
#Sta/Elev= 30
       0 3053.36     9.9 3051.07    69.6 3037.65    99.4 3030.23   109.3 3027.88
   119.3  3025.7   129.2 3023.67   139.2 3021.87   149.1 3020.26     159 3018.96
     169 3018.04   198.8 3015.92   208.7 3015.34   218.7 3015.01   248.5 3014.79
   308.1 3013.84   367.8 3013.21   407.5 3012.56   417.4  3012.3     424 3011.99
   427.4 3011.83   437.3  3011.1   447.3 3010.75   457.2 3011.74     4593012.118
   477.1 3016.03     487 3017.84   506.9  3021.1   516.8 3023.01   576.5 3035.69
#Mann= 3 , 0 , 0
       0      .1       0     424    .045       0     459      .1       0
Bank Sta=424,459
XS Rating Curve= 0 ,0
Exp/Cntr=0.3,0.1

Type RM Length L Ch R = 1 ,31142.2 ,211.5,211.8,212.2
XS GIS Cut Line= 2
     2114290.956      424696.206     2114867.009      424718.332
#Sta/Elev= 27
       0 3049.81    59.6 3035.25    89.4 3028.09    99.4 3025.81   119.3 3021.44
   139.2 3016.75   149.1 3014.66     169 3010.66   178.9 3009.14   188.8 3008.17
   208.7 3006.68   218.7 3006.06   228.6  3005.7   268.4 3005.54   298.2 3005.68
   304.93005.639     328 3005.52   337.9 3006.03   339.93006.348   347.9 3007.62
   357.8 3009.73   367.8 3011.72   417.4 3020.96   427.4  3022.7   437.3 3024.32
     487 3031.71   576.5 3044.71
#Mann= 3 , 0 , 0
       0      .1       0   304.9    .045       0   339.9      .1       0
Bank Sta=304.9,339.9
XS Rating Curve= 0 ,0
Exp/Cntr=0.3,0.1

Type RM Length L Ch R = 1 ,30930.4 ,331.4,329.1,326.8
XS GIS Cut Line= 2
     2114297.257      424898.849     2114751.706      424921.222
#Sta/Elev= 29
       0 3043.89     9.9  3041.2    19.8 3038.63    29.7 3036.22    39.6 3033.96
    59.4 3029.64    69.2  3027.4      89 3023.18    98.9 3021.25   108.8 3019.52
   118.7 3017.99   128.6 3016.68   138.5 3015.62   168.2 3013.21   207.7 3009.67
   227.5 3007.79   239.63006.456   247.3  3005.6   257.2 3004.89   267.1 3005.03
   274.63005.969     277 3006.27   286.8 3008.23   296.7 3010.05   306.6 3011.55
   336.3 3015.35   346.2 3016.86   435.2 3030.94     455 3033.95
#Mann= 3 , 0 , 0
       0      .1       0   239.6    .045       0   274.6      .1       0
Bank Sta=239.6,274.6
XS Rating Curve= 0 ,0
Exp/Cntr=0.3,0.1

Type RM Length L Ch R = 1 ,30601.3 ,139,136.7,134.4
XS GIS Cut Line= 2
     2114303.859      425243.216     2114758.191      425218.561
#Sta/Elev= 25
       0 3046.73    19.8 3041.23    39.6 3036.03    59.4 3031.06    79.1 3026.34
    98.9 3021.88   118.7 3017.62   138.5 3013.57   169.73007.383     178 3005.74
   187.9 3004.43   197.8  3004.1   204.73004.407   207.7 3004.54   227.5 3006.17
   267.1 3008.87     277 3009.66   286.8 3010.72   296.7 3012.05   336.3 3017.89
     366 3021.99   405.5 3027.21   415.4 3028.67   425.3 3030.46     455 3036.62
#Mann= 3 , 0 , 0
       0      .1       0   169.7    .045       0   204.7      .1       0
Bank Sta=169.7,204.7
XS Rating Curve= 0 ,0
Exp/Cntr=0.3,0.1

Type RM Length L Ch R = 1 ,30464.6 ,172.6,181.6,190.5
XS GIS Cut Line= 3
     2114354.996      425390.077     2114579.862      425355.556
     2114804.727      425321.035
#Sta/Elev= 25
       0 3035.82    29.7 3029.72    69.2 3021.86      89 3018.12   108.8 3014.48
   138.5 3009.27   148.4 3007.46   158.83005.425   168.2 3004.01     178 3003.58
   187.9 3004.08   193.8 3004.64   207.7 3005.91   237.4 3008.39   247.3 3009.32
   257.2 3010.63   267.1 3012.34   286.8 3016.06   316.5 3021.99   375.9 3034.34
   395.6 3038.32   405.5 3040.18   425.3 3043.72   435.2 3045.62     455  3049.7
#Mann= 3 , 0 , 0
       0      .1       0   158.8    .045       0   193.8      .1       0
Bank Sta=158.8,193.8
XS Rating Curve= 0 ,0
Exp/Cntr=0.3,0.1

Type RM Length L Ch R = 1 ,30283.1 ,257,273,288.9
XS GIS Cut Line= 3
     2114344.203      425497.758     2114661.502      425572.621
     2115035.444      425553.657
#Sta/Elev= 30
       0 3029.74    29.6  3024.6    59.3 3019.77    98.8  3013.7   148.2 3006.64
   163.8 3003.96     168 3003.26   177.8 3002.45   187.7 3002.28   198.83002.469
   207.5 3002.82   237.1 3004.79   276.6 3008.01   306.2 3010.26     326 3012.03
   335.9 3013.26   345.7 3014.94   355.6 3016.98     395 3025.59   454.1 3038.89
   523.1 3055.28   542.8 3059.69   562.5 3064.26   572.3 3066.41   641.3 3080.82
     661  3085.2   670.9  3087.6   680.7 3090.31   690.6  3093.5   700.4 3097.05
#Mann= 3 , 0 , 0
       0      .1       0   163.8    .045       0   198.8      .1       0
Bank Sta=163.8,198.8
XS Rating Curve= 0 ,0
Exp/Cntr=0.3,0.1

Type RM Length L Ch R = 1 ,30010.1 ,399.1,407.7,416.2
XS GIS Cut Line= 2
     2114201.368      425557.467     2114602.779      426101.074
#Sta/Elev= 30
       0 3033.05    20.2 3029.03    40.3 3025.31    60.5  3021.8    90.8 3016.89
   141.2 3008.99   151.3  3007.5   191.6 3002.54   201.7 3001.59   211.8 3001.36
   221.9  3001.8   226.63002.126   302.6 3007.79   342.9 3010.38   383.3 3012.54
   433.7 3014.52     474 3017.38   504.3 3019.77   524.5 3021.54   534.6 3022.62
   544.6 3023.87   554.7 3025.34     585 3030.38   605.2 3033.48   615.2 3034.78
   625.3 3035.87   645.5 3037.47   655.6 3038.81   665.7 3041.09   675.8 3043.93
#Mann= 3 , 0 , 0
       0      .1       0   191.6    .045       0   226.6      .1       0
Bank Sta=191.6,226.6
XS Rating Curve= 0 ,0
Exp/Cntr=0.3,0.1

Type RM Length L Ch R = 1 ,29602.4 ,283,288.4,293.9
XS GIS Cut Line= 2
     2113873.188      425601.986     2114020.197      426148.282
#Sta/Elev= 30
       0 3036.21    19.8 3032.68    39.7 3029.28    79.4 3022.74   109.2 3018.29
     129 3015.66   158.8 3012.05   188.6 3008.92   208.4 3007.08   248.1 3003.67
   265.4 3002.07   277.9 3001.06   287.8 3000.79   297.8 3001.18   300.43001.411
   317.6 3002.99   327.5 3003.72   377.2 3006.94   406.9 3009.53   436.7 3011.81
   446.6 3012.76   456.6 3013.88   466.5 3015.16   476.4 3016.82   486.3 3018.81
   496.3 3021.08   506.2 3023.63   516.1 3026.56   545.9 3036.06   565.7 3041.86
#Mann= 3 , 0 , 0
       0      .1       0   265.4    .045       0   300.4      .1       0
Bank Sta=265.4,300.4
XS Rating Curve= 0 ,0
Exp/Cntr=0.3,0.1

Type RM Length L Ch R = 1 ,29314   ,364.7,356.7,348.6
XS GIS Cut Line= 2
     2113710.913      425612.964     2113754.431      426177.019
#Sta/Elev= 30
       0 3033.23     9.9 3030.42    19.8 3028.06    29.8 3025.97    49.6 3022.15
    79.4 3017.22    99.2 3014.45   119.1    3012   148.9 3008.71   168.7  3006.9
   188.6 3005.55   198.5 3005.09   218.4 3004.52   297.8 3003.73   307.7 3003.76
   327.5 3004.15   357.3 3004.07   367.2  3003.8   377.2 3003.24   395.1 3001.53
   406.9  3000.6   416.8 3000.68   426.8  3002.2   430.1  3003.1   446.6 3007.45
   456.6  3009.6   476.4 3013.18   496.3 3016.18     536  3021.1   565.7 3025.12
#Mann= 3 , 0 , 0
       0      .1       0   395.1    .045       0   430.1      .1       0
Bank Sta=395.1,430.1
XS Rating Curve= 0 ,0
Exp/Cntr=0.3,0.1

Type RM Length L Ch R = 1 ,28957.4 ,316.3,313.4,311.7
XS GIS Cut Line= 2
     2113372.395      425656.443     2113589.804      426178.731
#Sta/Elev= 30
       0  3048.8    79.4 3032.84   109.2 3026.51   119.1 3024.16   168.7 3011.87
   178.6 3009.17   188.6 3005.91   198.5  3002.2   199.13002.042   208.4  2999.6
   218.4 3000.22   228.3  3003.1   234.13004.424   238.2 3005.36   248.1 3006.12
   307.7 3005.19   317.6 3004.69   327.5 3004.32   337.4 3004.15   347.4  3004.3
   367.2 3005.22   406.9 3007.49   416.8 3008.13   426.8 3008.91   436.7 3010.12
   516.1 3021.05     526 3022.26     536  3023.3   545.9 3024.05   565.7 3025.08
#Mann= 3 , 0 , 0
       0      .1       0   199.1    .045       0   234.1      .1       0
Bank Sta=199.1,234.1
XS Rating Curve= 0 ,0
Exp/Cntr=0.3,0.1

Type RM Length L Ch R = 1 ,28643.9 ,325.7,331.7,336.6
XS GIS Cut Line= 2
     2113180.371      425808.552     2113438.646      426311.886
#Sta/Elev= 30
       0 3024.99     9.9 3023.21    29.8 3019.94    79.4 3012.39    89.3 3011.02
    99.2 3009.94   109.2 3009.05     139 3006.74   158.8 3005.45   178.6 3004.68
   238.2 3003.07   277.9 3001.53   297.8 3000.24   317.6 2998.61   323.72998.456
   327.5 2998.36   337.4 2999.01   347.4 3000.51   358.73002.984   387.1 3009.24
   406.9 3013.87   416.8 3015.96   426.8 3017.72   436.7 3019.15   466.5 3022.83
   476.4 3024.17   496.3 3027.19     536 3033.77   555.8 3037.51   565.7 3039.56
#Mann= 3 , 0 , 0
       0      .1       0   323.7    .045       0   358.7      .1       0
Bank Sta=323.7,358.7
XS Rating Curve= 0 ,0
Exp/Cntr=0.3,0.1

Type RM Length L Ch R = 1 ,28312.2 ,220.8,222.1,223.3
XS GIS Cut Line= 2
     2112923.594      425846.692     2113082.045       426389.78
#Sta/Elev= 30
       0 3024.35    29.8 3019.25    49.6 3016.13    69.5 3013.24    89.3 3010.95
   109.2 3009.43     139  3007.7   208.4 3003.12   228.3 3002.39     258 3002.02
     268 3001.66   277.9 3000.67   287.8 2999.02   297.8 2997.56   299.52997.469
   307.7 2997.03   317.6 2997.24   334.52998.096   337.4 2998.26   347.4 2999.29
   357.3  3000.7   377.2 3003.92     397 3007.39   406.9 3008.85   426.8 3011.15
   476.4 3016.07   496.3 3018.39   506.2 3019.74     536 3024.66   565.7 3030.16
#Mann= 3 , 0 , 0
       0      .1       0   299.5    .045       0   334.5      .1       0
Bank Sta=299.5,334.5
XS Rating Curve= 0 ,0
Exp/Cntr=0.3,0.1

Type RM Length L Ch R = 1 ,28090.2 ,489.7,485.8,480.4
XS GIS Cut Line= 2
     2112729.287      425905.834     2112857.064       426451.87
#Sta/Elev= 30
       0 3015.57      20 3012.67    70.1 3006.45    80.1  3005.4    90.1  3004.7
   100.1 3004.39   110.2 3004.33   160.2 3004.84   180.2 3005.16   190.3 3005.18
   200.3 3004.76   210.3 3003.97   220.3 3002.87   230.3 3001.54   250.4 2998.62
   260.4 2997.47   262.92997.337   270.4 2996.94   280.4 2997.17   297.92998.657
   310.4 2999.68   360.5 3002.98   380.5 3004.45   400.6 3006.31   430.6 3009.69
   470.7 3015.07   490.7 3018.33   520.7 3023.65   540.8 3027.61   560.8 3031.82
#Mann= 3 , 0 , 0
       0      .1       0   262.9    .045       0   297.9      .1       0
Bank Sta=262.9,297.9
XS Rating Curve= 0 ,0
Exp/Cntr=0.3,0.1

Type RM Length L Ch R = 1 ,27604.4 ,491.1,485.4,475.3
XS GIS Cut Line= 2
     2112240.423      426012.394     2112425.616      426541.719
#Sta/Elev= 30
       0 3033.71      20 3028.76      30 3026.49    50.1 3022.33    60.1  3020.4
    70.1 3018.67    80.1 3017.04    90.1 3015.53   100.1 3014.13   120.2 3011.43
   140.2 3008.37   160.2 3005.12   170.2 3003.62   180.2 3002.31   190.3  3001.2
   200.3 3000.24   210.3 2999.36   224.12998.285   240.3 2997.19   250.4 2996.75
   259.12996.541   280.4 2996.41   340.5 2996.42   370.5 2996.55   380.5 2996.65
   390.6 2996.94   400.6 2997.58   410.6 2998.65   450.6 3003.36   560.8 3016.66
#Mann= 3 , 0 , 0
       0      .1       0   224.1    .045       0   259.1      .1       0
Bank Sta=224.1,259.1
XS Rating Curve= 0 ,0
Exp/Cntr=0.3,0.1

Type RM Length L Ch R = 1 ,27119   ,829.3,817,818.3
XS GIS Cut Line= 3
     2111840.248      426023.605     2111897.851      426221.395
     2112218.089      426746.384
#Sta/Elev= 30
       0 3032.96    19.6 3029.13      49 3024.17    68.7 3021.08    98.1 3017.01
   117.7 3014.64   137.3 3012.53     157 3010.73   186.4 3008.35   246.3  3004.4
   296.7 3001.55   316.9 3000.84   377.4 2999.66   508.4 2995.93   508.9 2995.93
   518.5 2995.93   528.6 2996.27   543.92997.427   548.8  2997.8   558.8 2998.23
   568.9 2998.44   629.4 2998.77   649.6 2999.16   679.8 3000.54   720.2 3002.92
   730.2 3003.64   740.3 3004.57   760.5 3006.72   790.7 3010.29     821 3014.18
#Mann= 3 , 0 , 0
       0      .1       0   508.9    .045       0   543.9      .1       0
Bank Sta=508.9,543.9
XS Rating Curve= 0 ,0
Exp/Cntr=0.3,0.1

Type RM Length L Ch R = 1 ,26302   ,283.7,282.5,281.3
XS GIS Cut Line= 2
     2111340.715      426636.841      2111823.78      426921.674
#Sta/Elev= 27
       0 3026.85      10 3023.38      20 3020.11      30 3017.09    40.1 3014.31
    50.1 3011.76    60.1 3009.39    70.1  3007.3    80.1 3005.42    90.1 3003.92
   120.2 2999.64   140.2 2997.13   150.2 2996.22   160.2  2995.7   180.2 2995.06
   190.3 2994.96   200.3 2995.02   220.3 2995.52   232.72995.665   260.4 2995.63
   267.72995.747   290.4  2996.4   300.4  2996.6   440.6 2998.47   470.7 2999.21
   540.8 3001.48   560.8 3001.89
#Mann= 3 , 0 , 0
       0      .1       0   232.7    .045       0   267.7      .1       0
Bank Sta=232.7,267.7
XS Rating Curve= 0 ,0
Exp/Cntr=0.3,0.1

Type RM Length L Ch R = 1 ,26019.5 ,569.5,541.9,535.1
XS GIS Cut Line= 2
     2111187.081      426877.588     2111813.354       427206.31
#Sta/Elev= 30
       0 3033.52    39.8 3022.25    59.8 3016.94    69.7 3014.51    79.7 3012.34
    89.7 3010.44    99.6 3008.82   119.5 3006.06   139.5 3003.62   149.4 3002.55
   169.4 3000.81   199.2 2999.02   239.1 2997.28   258.92995.888   268.9 2995.25
   278.9    2995   293.9 2995.07   328.8 2995.36   398.5 2994.54   448.3  2994.3
   458.2 2994.32   468.2  2994.6     528 2997.79   557.9 2999.66   587.8 3002.05
   607.7 3004.14   617.6 3005.55   647.5 3010.38   667.4  3013.4   707.3 3018.99
#Mann= 3 , 0 , 0
       0      .1       0   258.9    .045       0   293.9      .1       0
Bank Sta=258.9,293.9
XS Rating Curve= 0 ,0
Exp/Cntr=0.3,0.1

Type RM Length L Ch R = 1 ,25477.7 ,615.9,606.9,597.5
XS GIS Cut Line= 2
     2110960.649      427219.868     2111629.495      427449.913
#Sta/Elev= 30
       0 3010.28      10 3008.93    19.9  3007.9    29.9 3007.28    39.8 3007.13
    49.8 3007.42    59.8 3007.52    69.7 3007.06    79.7 3006.26    89.7  3005.2
   109.6 3002.81   129.5 3000.78   169.4 2997.46   189.3 2996.12   209.2 2995.18
     249 2993.72   286.1 2992.72   308.8 2992.17   318.8 2992.09   321.12992.095
   338.7  2992.2   378.6 2992.85     518 2996.13     528 2996.47   567.8  2998.9
   627.6 3002.27   647.5 3003.77   657.5 3004.81   677.4 3007.35   707.3 3011.84
#Mann= 3 , 0 , 0
       0      .1       0   286.1    .045       0   321.1      .1       0
Bank Sta=286.1,321.1
XS Rating Curve= 0 ,0
Exp/Cntr=0.3,0.1

Type RM Length L Ch R = 1 ,24870.8 ,533.9,533.7,531.9
XS GIS Cut Line= 2
     2110934.362      427896.297     2111663.237      427834.559
#Sta/Elev= 30
       0 3018.28      20 3013.27    40.1 3008.71    60.1 3004.57    70.1 3002.72
    80.2 3001.06    90.2 2999.65   100.2 2998.42   120.2 2996.47   140.3 2995.46
   200.4  2993.5   240.5 2992.46   310.6 2991.43   364.32991.038   380.8 2990.86
   390.8 2990.88   399.3 2991.22   420.8 2992.68   460.9 2994.88     481 2995.42
   551.1 2996.31   591.2 2997.78   611.2 2998.83   621.3 2999.55   631.3 3000.59
   641.3 3001.97   661.3 3005.17   701.4 3011.94   711.4  3013.5   731.5 3016.23
#Mann= 3 , 0 , 0
       0      .1       0   364.3    .045       0   399.3      .1       0
Bank Sta=364.3,399.3
XS Rating Curve= 0 ,0
Exp/Cntr=0.3,0.1

Type RM Length L Ch R = 1 ,24337.1 ,361.8,359.5,360.7
XS GIS Cut Line= 2
     2110969.881      428341.484     2111713.163      428292.971
#Sta/Elev= 30
       0 3009.19    30.2 3005.49    50.3 3003.51    80.5 3000.77   100.7 2999.29
   130.8 2997.45   191.2 2993.25   201.3 2992.86     312 2990.67   371.52989.789
   406.52989.546   412.7 2989.54   422.8 2989.58   442.9 2989.94   483.2 2991.22
   493.2 2991.95   503.3 2993.11   513.4 2994.78   543.6 3000.94   553.6 3003.11
   583.8    3010   603.9 3014.26   654.3 3023.97   664.3  3025.7   684.5 3028.88
   694.5 3031.08   704.6 3033.64   714.7 3036.37   724.7 3039.36   744.9 3045.97
#Mann= 3 , 0 , 0
       0      .1       0   371.5    .045       0   406.5      .1       0
Bank Sta=371.5,406.5
XS Rating Curve= 0 ,0
Exp/Cntr=0.3,0.1

Type RM Length L Ch R = 1 ,23977.6 ,416.1,417.3,418.4
XS GIS Cut Line= 3
     2111037.105       428610.99     2111389.972      428579.729
     2111615.386      428560.945
#Sta/Elev= 23
       0 3002.55    19.7  3001.3    49.2 2999.25    98.4 2996.29   177.1  2991.4
     187 2990.82   196.8 2990.38   216.5 2989.97   369.12988.018   393.6  2987.7
   404.12987.911   413.3 2988.45   423.1 2989.37   432.9 2990.44   442.8 2991.83
   472.3  2996.9   482.1 2998.74   491.9 3000.73   501.8 3002.92   531.3 3009.96
   541.1 3012.42   560.8  3017.7   580.4 3023.36
#Mann= 3 , 0 , 0
       0      .1       0   369.1    .045       0   404.1      .1       0
Bank Sta=369.1,404.1
XS Rating Curve= 0 ,0
Exp/Cntr=0.3,0.1

Type RM Length L Ch R = 1 ,23560.3 ,580.8,569.3,557.4
XS GIS Cut Line= 2
     2110747.122      428969.668     2111844.971      428982.149
#Sta/Elev= 30
       0 3029.16   110.8 3007.95   130.9 3004.36   171.2 2998.37   191.4 2996.79
     272 2993.06   332.4 2991.34   513.7    2988     671 2987.09     695 2987.02
     7062987.067   725.2 2987.68   765.5 2989.78   775.6 2990.65   785.7  2992.6
   805.8  2999.7   815.9 3002.78     826 3005.13     836 3006.93   846.1 3008.09
   866.2 3009.58   876.3 3011.29   906.5 3017.58   936.8 3024.49     967 3032.44
   997.2 3041.71  1027.4 3051.91  1057.6 3061.28  1077.8 3067.06  1097.9 3072.11
#Mann= 3 , 0 , 0
       0      .1       0     671    .045       0     706      .1       0
Bank Sta=671,706
XS Rating Curve= 0 ,0
Exp/Cntr=0.3,0.1

Type RM Length L Ch R = 1 ,22991   ,469.2,482.7,494.7
XS GIS Cut Line= 3
     2110667.244      429675.284     2111176.891      429532.174
     2112210.013      429304.116
#Sta/Elev= 30
       0 3030.72    89.9 3016.18   119.8 3011.54   169.8 3004.77   189.8 3002.58
   199.8 3001.76   289.6 2995.94   309.6  2995.1   339.6 2994.42   469.4 2993.19
   499.4 2992.69   539.4 2991.76   589.8 2990.04   690.6 2987.98   831.12987.371
   866.12987.243   932.4 2986.99  1002.9 2987.03  1063.4 2987.63  1073.5 2988.09
  1083.6 2988.91  1123.8 2992.74    1144 2993.99  1264.9  2997.6  1295.1 2998.68
  1315.3  2999.7  1416.1 3008.43  1456.4 3012.45    1537 3023.24  1587.4 3029.56
#Mann= 3 , 0 , 0
       0      .1       0   831.1    .045       0   866.1      .1       0
Bank Sta=831.1,866.1
XS Rating Curve= 0 ,0
Exp/Cntr=0.3,0.1

Type RM Length L Ch R = 1 ,22508.3 ,489.6,488.4,487.9
XS GIS Cut Line= 3
     2110642.974      429734.857     2111161.366      429662.733
     2112102.505      429815.391
#Sta/Elev= 30
       0 3032.88    50.3 3024.85    80.5 3020.25     151 3010.11     161 3008.89
   181.2 3007.03   221.4 3004.65   261.7 3003.09   402.6 2997.05   543.5 2993.47
   653.9 2989.19     684  2988.2   754.2 2987.01   874.6 2985.86   914.8 2984.76
   954.9 2984.91  1105.5 2983.92  1109.22983.927  1125.6 2984.12  1144.22985.301
  1195.8 2988.65    1246 2991.34    1256 2992.28  1286.1 2995.74  1326.3 3000.74
  1356.4 3004.76  1406.6 3012.25  1436.7  3017.6  1456.8  3021.5  1476.8 3025.66
#Mann= 3 , 0 , 0
       0      .1       0  1109.2    .045       0  1144.2      .1       0
Bank Sta=1109.2,1144.2
XS Rating Curve= 0 ,0
Exp/Cntr=0.3,0.1

Type RM Length L Ch R = 1 ,22019.9 ,346.1,346.1,345.1
XS GIS Cut Line= 2
     2110631.942       429873.86     2112033.004      430101.119
#Sta/Elev= 30
       0 3032.03    20.1 3028.27    50.3 3023.26    70.5 3020.49   100.7 3017.74
   140.9  3012.4   261.7  3000.1   291.9 2997.41   322.1 2993.51   342.3 2991.55
   372.5  2989.6   392.6 2988.78     453 2988.04   563.7 2984.11   583.9 2983.89
   704.6 2983.89   739.82984.384   774.82984.473   805.3  2983.9   946.2  2983.9
  1026.8 2984.63    1067 2985.47  1127.4  2989.2  1177.8 2994.06    1208 2997.35
  1258.3 3003.63  1278.4 3006.65  1308.6 3012.28    1359 3023.86  1419.4 3036.37
#Mann= 3 , 0 , 0
       0      .1       0   739.8    .045       0   774.8      .1       0
Bank Sta=739.8,774.8
XS Rating Curve= 0 ,0
Exp/Cntr=0.3,0.1

Type RM Length L Ch R = 1 ,21673.8 ,565.8,568.5,571.2
XS GIS Cut Line= 2
     2110774.468      430268.451     2112119.053      430370.299
#Sta/Elev= 30
       0 3019.57    40.2 3014.53   120.8 3005.82   191.2 2997.12   221.4 2993.84
   261.6 2990.31   301.9 2987.81   352.2 2985.61   412.6  2984.9   442.8    2984
   462.9 2983.89   477.1 2983.89   512.1 2983.89   553.5  2983.9   603.8 2984.82
   774.8 2985.18     805 2985.83   875.5 2989.14   895.6 2990.75   996.2 3002.93
  1016.4 3005.76  1096.9 3019.92    1117 3024.57  1177.4  3039.9  1237.8 3052.51
  1257.9 3057.17    1278 3063.22  1288.1 3066.83  1318.2    3079  1348.4 3090.33
#Mann= 3 , 0 , 0
       0      .1       0   477.1    .045       0   512.1      .1       0
Bank Sta=477.1,512.1
XS Rating Curve= 0 ,0
Exp/Cntr=0.3,0.1

Type RM Length L Ch R = 1 ,21105.2 ,450.4,455.4,453
XS GIS Cut Line= 2
     2110786.377      430743.381     2112127.879      431021.187
#Sta/Elev= 30
       0  3006.7    10.1 3004.61    20.2 3003.21   100.7 2995.38   120.9 2993.76
     141 2992.47   181.3 2990.48   211.5 2989.55   241.8    2989     272 2988.93
   362.6 2989.38     413 2988.93   443.2 2988.27   453.3 2987.88   503.7  2985.1
   526.72984.042     544 2983.89   561.72983.897   584.2 2984.18   614.5 2984.98
   765.6 2990.05   815.9 2991.56   856.2 2992.57   886.4 2993.09   936.8 2993.54
  1027.5 2994.72  1148.4 2996.71    1239 2998.97  1339.8    3001    1370 3001.74
#Mann= 3 , 0 , 0
       0      .1       0   526.7    .045       0   561.7      .1       0
Bank Sta=526.7,561.7
XS Rating Curve= 0 ,0
Exp/Cntr=0.3,0.1

Type RM Length L Ch R = 1 ,20649.8 ,438.5,439,439.5
XS GIS Cut Line= 2
        2110615.      430862.984     2111617.685      431294.254
#Sta/Elev= 30
       0 3017.32      10 3014.56      20 3012.16      30 3010.08    40.1 3008.35
    50.1 3007.26    80.1 3005.27   220.3 2995.42   250.3 2993.56   260.4 2993.07
   280.4 2992.48   340.5 2992.52   420.6 2991.16   470.6 2989.88   580.8 2986.53
   650.9 2984.94     731 2983.95   774.22983.951   791.1  2983.9   801.1 2983.96
   809.22984.397   811.1  2984.5   831.1 2987.14   861.2 2990.63   961.3 3001.72
   991.4 3004.84  1001.4 3005.63  1011.4 3006.09  1051.4 3007.12  1091.5 3007.72
#Mann= 3 , 0 , 0
       0      .1       0   774.2    .045       0   809.2      .1       0
Bank Sta=774.2,809.2
XS Rating Curve= 0 ,0
Exp/Cntr=0.3,0.1

Type RM Length L Ch R = 1 ,20210.8 ,207.3,207.3,207.3
XS GIS Cut Line= 2
     2110842.316      431370.661     2111259.413      431552.472
#Sta/Elev= 20
       0 2994.47    49.5 2992.24   108.8 2989.27   148.4 2986.91     178 2984.78
   187.9 2984.42   235.22983.913   245.2 2983.89   270.22983.912     277 2983.96
   286.8 2984.83   306.6 2988.41   316.5 2990.04   356.1 2996.33     366 2997.72
   375.9  2998.5   385.8 2998.74   435.2 2999.12   445.1 2999.61     455 3000.82
#Mann= 3 , 0 , 0
       0      .1       0   235.2    .045       0   270.2      .1       0
Bank Sta=235.2,270.2
XS Rating Curve= 0 ,0
Exp/Cntr=0.3,0.1

Type RM Length L Ch R = 1 ,20003.6 ,190.5,194.8,199.1
XS GIS Cut Line= 3
     2110794.765      431573.067     2111003.314      431663.973
     2111211.862      431754.878
#Sta/Elev= 25
       0 2994.05    69.2 2989.93   118.7 2987.21     178 2984.36   187.9    2984
   197.8  2983.9   199.62983.902   234.62983.946   237.4 2983.96   247.3 2984.48
   257.2 2985.69     277 2988.58   306.6 2992.42   326.4 2994.39   336.3 2995.25
   346.2 2995.99   356.1 2996.59     366 2996.95   385.8 2997.26   395.6 2997.54
   405.5 2998.23   425.3 2999.98   435.2 3000.98   445.1 3002.25     455 3003.86
#Mann= 3 , 0 , 0
       0      .1       0   199.6    .045       0   234.6      .1       0
Bank Sta=199.6,234.6
XS Rating Curve= 0 ,0
Exp/Cntr=0.3,0.1

Type RM Length L Ch R = 1 ,19808.7 ,206.2,209.6,213.1
XS GIS Cut Line= 2
     2110735.514      431719.031     2111111.281      431975.593
#Sta/Elev= 19
       0 2995.73    29.7 2993.92   138.5  2986.8   158.3  2985.4   168.2 2984.52
   170.52984.405     178 2984.03   187.9  2983.9   197.8 2983.99   205.52984.395
   207.7 2984.51   217.6 2985.63   227.5 2986.54   336.3 2995.65   346.2 2996.53
   356.1 2997.58     366 2998.95   425.3 3009.13     455 3014.32
#Mann= 3 , 0 , 0
       0      .1       0   170.5    .045       0   205.5      .1       0
Bank Sta=170.5,205.5
XS Rating Curve= 0 ,0
Exp/Cntr=0.3,0.1

Type RM Length L Ch R = 1 ,19599.1 ,466.1,458.5,450.8
XS GIS Cut Line= 2
     2110616.455      431855.069     2110949.021      432165.592
#Sta/Elev= 29
       0 3012.77     9.9 3009.85    19.8 3007.12    29.7 3004.55    39.6 3002.16
    49.5 2999.92    59.4 2997.79    69.2 2995.91    79.1 2994.68    98.9 2994.47
   108.8 2993.86   118.7 2992.91   128.6 2991.58   138.5  2990.1   148.4 2988.49
   168.2 2985.03   170.32984.822     178 2984.06   187.9 2983.89   197.8 2983.98
   205.32984.359   227.5 2985.92   326.4 2991.79   356.1  2993.6     366 2994.31
   375.9 2995.29   385.8 2996.39   405.5 2998.76     455 3005.18
#Mann= 3 , 0 , 0
       0      .1       0   170.3    .045       0   205.3      .1       0
Bank Sta=170.3,205.3
XS Rating Curve= 0 ,0
Exp/Cntr=0.3,0.1

Type RM Length L Ch R = 1 ,19140.6 ,175.2,176.2,177.3
XS GIS Cut Line= 2
     2110296.597      432278.066     2110713.694      432459.877
#Sta/Elev= 23
       0 3027.34    59.4 3010.07    69.2 3007.11      89 3000.79    98.9 2997.84
   108.8  2995.4   118.7 2993.61   128.6 2992.31   138.5 2991.24   148.4 2990.29
   168.2 2988.74   207.7 2986.22   233.12984.368   237.4 2984.06   247.3 2983.67
   257.2 2983.88   268.12984.834   286.8 2986.72   375.9 2994.75   385.8 2995.88
   395.6  2997.3   415.4 3000.37     455 3006.78
#Mann= 3 , 0 , 0
       0      .1       0   233.1    .045       0   268.1      .1       0
Bank Sta=233.1,268.1
XS Rating Curve= 0 ,0
Exp/Cntr=0.3,0.1

Type RM Length L Ch R = 1 ,18964.4 ,460.5,465.7,470.9
XS GIS Cut Line= 2
     2110250.922      432437.542      2110666.68      432642.515
#Sta/Elev= 30
       0 3018.07    10.1 3014.88    20.2 3012.24    30.2 3009.76    40.3 3007.37
    50.4 3005.07    60.5 3002.89    70.5 3000.88    90.7 2997.18   100.8  2995.5
   110.8 2993.94     131 2991.12   161.2 2987.26   201.5 2982.43   214.32980.609
   221.7 2979.51   231.8 2978.71   241.8  2979.1   249.32979.984     262  2981.6
   272.1 2982.76   302.3  2986.1   352.7 2991.54   362.8 2992.71   382.9 2995.23
     393 2996.74   403.1 2998.48   413.2 3000.43   433.3 3004.64   463.5 3011.13
#Mann= 3 , 0 , 0
       0      .1       0   214.3    .045       0   249.3      .1       0
Bank Sta=214.3,249.3
XS Rating Curve= 0 ,0
Exp/Cntr=0.3,0.1

Type RM Length L Ch R = 1 ,18498.7 ,471.2,478.7,486.2
XS GIS Cut Line= 2
     2110156.305      432791.357     2110511.821      433088.808
#Sta/Elev= 30
       0 3024.27    50.4 3011.73    70.5 3006.88   110.8 2997.46   161.2 2986.33
   201.5 2978.14   214.32975.239   221.7 2973.73   231.8 2972.95   241.8 2974.03
   249.32976.325   251.9 2977.12     262 2980.54   272.1 2983.69   282.2 2986.56
   292.2  2988.4   302.3 2989.09   312.4 2990.09   322.5 2991.93   332.5 2995.04
   352.7 3002.45   362.8 3006.56   382.9 3015.73     393  3019.5   403.1 3023.04
   413.2 3026.46   423.2 3029.69   433.3  3032.8   453.5  3038.4   463.5 3041.02
#Mann= 3 , 0 , 0
       0      .1       0   214.3    .045       0   249.3      .1       0
Bank Sta=214.3,249.3
XS Rating Curve= 0 ,0
Exp/Cntr=0.3,0.1

Type RM Length L Ch R = 1 ,18020   ,522.2,517.3,512.4
XS GIS Cut Line= 2
     2109840.336      433041.388     2110080.187       433438.05
#Sta/Elev= 30
       0 3046.11    20.2  3038.4    40.3 3030.22    90.7 3008.69   110.8 3000.26
     131 2992.19   151.2 2984.35   171.3 2976.28   181.4 2972.03   183.92971.258
   191.5 2968.91   201.5 2967.87   211.6 2969.01   218.92970.817   231.8 2974.24
   241.8 2976.65     262 2981.34   272.1 2983.22   282.2 2984.29   302.3 2985.29
   312.4 2986.01   322.5 2987.03   332.5 2988.34   342.6 2989.96   352.7 2991.88
   362.8    2994   372.8 2996.34   382.9 2998.89   413.2 3006.99   463.5 3019.59
#Mann= 3 , 0 , 0
       0      .1       0   183.9    .045       0   218.9      .1       0
Bank Sta=183.9,218.9
XS Rating Curve= 0 ,0
Exp/Cntr=0.3,0.1

Type RM Length L Ch R = 1 ,17502.7 ,501.1,501.4,520.6
XS GIS Cut Line= 2
     2109373.556      433357.123     2109687.482      433686.479
#Sta/Elev= 30
       0 3029.59    29.7 3018.13    39.6 3014.56    49.5 3011.37    69.2  3006.6
    79.1 3003.84   158.3 2978.37   187.9 2969.09   197.8 2966.09   207.7  2962.9
   216.1 2959.99   217.6 2959.47   227.5 2956.76   237.4 2956.57   247.3 2959.43
   251.12961.779   257.2 2965.55   267.1  2972.3     277 2977.88   286.8 2982.17
   296.7 2984.99   316.5 2989.51   346.2 2996.07   356.1  2998.7     366 3002.06
   375.9 3005.91   415.4 3022.19   435.2 3030.22   445.1 3034.02     455 3037.18
#Mann= 3 , 0 , 0
       0      .1       0   216.1    .045       0   251.1      .1       0
Bank Sta=216.1,251.1
XS Rating Curve= 0 ,0
Exp/Cntr=0.3,0.1

Type RM Length L Ch R = 1 ,17001.3 ,241.9,238.6,235.5
XS GIS Cut Line= 3
     2109011.626      433702.097     2109168.589      433866.775
     2109325.552      434031.453
#Sta/Elev= 30
       0 3011.77    19.8  3006.5    59.4 2995.35    69.2 2992.84      89 2988.29
   108.8 2984.72   118.7 2982.51   158.3 2972.35   197.8 2962.43     2102959.096
   217.6  2957.2   227.5 2955.75   237.4 2957.26     2452960.914   247.3 2962.02
   257.2 2968.33   267.1 2973.43     277 2976.59   306.6 2983.43   316.5 2985.57
   326.4 2987.63   346.2 2991.22     366  2994.3   375.9  2995.4   395.6 2996.91
   405.5 2998.03   415.4 2999.94   425.3 3002.43   435.2 3005.12     455 3010.88
#Mann= 3 , 0 , 0
       0      .1       0     210    .045       0     245      .1       0
Bank Sta=210,245
XS Rating Curve= 0 ,0
Exp/Cntr=0.3,0.1

Type RM Length L Ch R = 1 ,16762.7 ,260.3,281.5,302.7
XS GIS Cut Line= 2
     2108833.153      433903.272     2109190.556      434184.854
#Sta/Elev= 30
       0 2999.93    19.8 2997.52    39.6 2995.26    69.2 2992.19    79.1 2990.84
      89  2988.5    98.9  2985.5   118.7 2979.17   148.4 2969.34     178 2959.78
   187.9 2956.35   190.72955.578   197.8 2953.62   207.7  2952.8   217.6 2953.68
   225.72955.218   237.4 2957.59   257.2 2961.13   286.8 2966.19   296.7 2967.58
   306.6 2968.59   316.5 2969.38   326.4 2969.83   336.3 2970.55   405.5 2976.06
   415.4 2976.95   425.3  2978.1   435.2 2979.05   445.1 2979.34     455  2978.9
#Mann= 3 , 0 , 0
       0      .1       0   190.7    .045       0   225.7      .1       0
Bank Sta=190.7,225.7
XS Rating Curve= 0 ,0
Exp/Cntr=0.3,0.1

Type RM Length L Ch R = 1 ,16481.2 ,336.1,350.2,365.3
XS GIS Cut Line= 2
      2108819.77       433912.69     2108808.202      434367.543
#Sta/Elev= 30
       0 2997.05     9.9 2994.56    19.8 2992.17    29.7 2990.06    39.6 2988.18
    69.2 2982.96   108.8 2976.66   118.7 2975.02   138.5 2971.54   148.4 2969.97
   158.3 2968.54   168.2 2967.32     178 2966.42   187.9 2965.81   207.7 2964.85
   217.6  2964.2   227.5 2963.28   237.4 2962.06   267.1 2957.77     277  2956.2
   290.62953.709   296.7  2952.6   306.6 2951.92   316.5 2952.13   325.62954.364
   326.4 2954.56   336.3 2958.42   346.2 2961.68   356.1 2964.32     455 2989.74
#Mann= 3 , 0 , 0
       0      .1       0   290.6    .045       0   325.6      .1       0
Bank Sta=290.6,325.6
XS Rating Curve= 0 ,0
Exp/Cntr=0.3,0.1

Type RM Length L Ch R = 1 ,16131   ,141.9,127.4,112.9
XS GIS Cut Line= 2
     2108745.374      433766.971     2108482.472      434138.331
#Sta/Elev= 28
       0 3023.42    39.6 3018.32    49.5 3016.83    59.4 3014.71    69.2 3011.48
    98.9    3001   158.3 2981.35   187.9 2971.76   217.6 2962.69   227.5 2959.82
   237.4 2957.67   247.3  2956.2   257.2 2954.94   267.1 2952.93   275.22950.647
     277 2950.14   286.8 2948.19   296.7 2947.91   310.2 2949.26   316.5 2949.89
   326.4 2950.17   336.3 2950.26   346.2 2950.83   356.1 2952.59   385.8 2959.27
   405.5 2963.64   435.2 2970.09     455 2974.56
#Mann= 3 , 0 , 0
       0      .1       0   275.2    .045       0   310.2      .1       0
Bank Sta=275.2,310.2
XS Rating Curve= 0 ,0
Exp/Cntr=0.3,0.1

Type RM Length L Ch R = 1 ,16003.6 ,233.2,242.2,251.1
XS GIS Cut Line= 2
     2108458.911      433723.726     2108467.218       434178.65
#Sta/Elev= 30
       0 3017.78     9.9 3014.34    79.1  2989.7   108.8 2978.85   118.7  2975.3
   128.6 2971.84   148.4 2965.07   158.3 2961.84   168.2 2958.84   197.8 2950.42
   216.6 2944.64   217.6 2944.33   227.5  2942.2   237.4 2941.84   247.3 2942.78
   251.62943.292   257.2 2943.96   267.1 2944.82   286.8    2946   296.7 2946.99
   306.6 2948.86   316.5 2951.61   336.3 2957.36   346.2 2959.97   356.1 2962.42
   375.9 2967.04   415.4 2976.01   435.2 2980.28   445.1 2982.29     455 2984.49
#Mann= 3 , 0 , 0
       0      .1       0   216.6    .045       0   251.6      .1       0
Bank Sta=216.6,251.6
XS Rating Curve= 0 ,0
Exp/Cntr=0.3,0.1

Type RM Length L Ch R = 1 ,15761.5 ,272.1,269.5,266.9
XS GIS Cut Line= 2
      2108320.66      433690.771     2108153.782      434114.064
#Sta/Elev= 30
       0 3003.95     9.9    3000    19.8 2996.28    29.7 2992.74    98.9  2968.5
   128.6 2957.93   138.5 2954.57   148.4 2951.77   158.3 2949.66   187.9 2944.35
   217.6 2939.24   227.5 2937.21   234.62935.482   237.4  2934.8   247.3 2932.82
   257.2 2932.35   267.1 2934.06   269.62935.075     277 2938.08   286.8 2942.76
   296.7 2946.24   326.4 2955.47   346.2 2961.25   385.8  2972.5   395.6 2975.38
   405.5  2978.4   415.4 2981.76   425.3 2985.97   435.2 2990.74     455 3000.58
#Mann= 3 , 0 , 0
       0      .1       0   234.6    .045       0   269.6      .1       0
Bank Sta=234.6,269.6
XS Rating Curve= 0 ,0
Exp/Cntr=0.3,0.1

Type RM Length L Ch R = 1 ,15492   ,219.1,212.3,205.4
XS GIS Cut Line= 3
     2108038.752      433602.311     2107980.016      433822.098
      2107921.28      434041.885
#Sta/Elev= 28
       0 2989.73     9.9 2986.78    29.7 2980.69    39.6 2977.57    49.5 2974.33
    98.9 2957.23   118.7 2950.71   138.5 2944.38     178 2931.95   187.9 2929.22
   197.8 2926.29   207.7 2922.88     2102922.229   217.6 2920.08   227.5 2918.87
   237.4  2919.5     2452921.358   247.3 2921.92   257.2 2925.07   267.1  2927.8
     277 2930.29   296.7 2935.58   306.6 2938.32   316.5 2941.17   326.4 2944.12
   385.8 2962.33   425.3 2974.79     455 2984.02
#Mann= 3 , 0 , 0
       0      .1       0     210    .045       0     245      .1       0
Bank Sta=210,245
XS Rating Curve= 0 ,0
Exp/Cntr=0.3,0.1

Type RM Length L Ch R = 1 ,15279.7 ,236.8,230.9,225
XS GIS Cut Line= 2
     2107765.183      433594.329     2107783.591      434048.957
#Sta/Elev= 30
       0    2953    19.8 2948.21    39.6 2942.11    49.5 2939.51    79.1 2933.48
   108.8 2928.96   118.7 2927.02   128.6  2924.7   158.3  2916.8   168.2 2914.01
   175.62911.533   187.9 2908.38   197.8 2907.71   207.7  2908.6   210.62909.265
   217.6 2910.87   237.4 2916.39   267.1 2923.14     277 2925.84   286.8 2929.01
   306.6 2935.93   326.4  2943.4   336.3 2947.54     366 2961.12   395.6 2974.19
   405.5 2978.12   415.4 2981.39   425.3 2983.82   445.1 2986.94     455 2989.35
#Mann= 3 , 0 , 0
       0      .1       0   175.6    .045       0   210.6      .1       0
Bank Sta=175.6,210.6
XS Rating Curve= 0 ,0
Exp/Cntr=0.3,0.1

Type RM Length L Ch R = 1 ,15048.8 ,271.1,257.4,243.7
XS GIS Cut Line= 2
     2107484.031       433628.18     2107620.224      434062.318
#Sta/Elev= 30
       0 2933.68    29.7 2924.49    39.6 2922.22    49.5 2921.22    59.4  2921.1
    79.1 2921.35      89 2920.68    98.9 2919.18   158.3 2907.84   168.2 2905.83
     178 2903.44   188.32900.623   197.8 2899.02   207.7 2899.01   217.6 2900.91
   223.32902.695   237.4 2906.79   247.3 2908.85   257.2 2910.46     277 2913.08
   286.8 2914.73   296.7 2917.09   306.6  2920.5   336.3 2932.31   375.9 2948.35
   395.6 2957.54   405.5 2961.24   415.4 2963.94   425.3 2965.99     455 2971.67
#Mann= 3 , 0 , 0
       0      .1       0   188.3    .045       0   223.3      .1       0
Bank Sta=188.3,223.3
XS Rating Curve= 0 ,0
Exp/Cntr=0.3,0.1

Type RM Length L Ch R = 1 ,14791.4 ,263.4,257.9,252.5
XS GIS Cut Line= 2
     2107202.443      433839.921     2107558.787      434122.841
#Sta/Elev= 28
       0 2944.91    19.8 2937.47    39.6 2929.84    49.5  2925.9    59.4 2921.79
   108.8 2899.44   118.7 2894.04     1242891.823   128.6  2889.9   138.5 2888.15
   148.4 2889.08     1592891.223   168.2 2893.23     178  2894.7   187.9 2895.77
   217.6 2898.67   227.5 2899.42   237.4 2899.47   267.1 2898.48     277  2898.6
   286.8 2899.93   296.7 2902.76   326.4  2912.8     366 2926.62   385.8 2933.76
   395.6 2937.37   425.3    2948     455 2958.95
#Mann= 3 , 0 , 0
       0      .1       0     124    .045       0     159      .1       0
Bank Sta=124,159
XS Rating Curve= 0 ,0
Exp/Cntr=0.3,0.1

Type RM Length L Ch R = 1 ,14533.5 ,245.2,256.9,285.9
XS GIS Cut Line= 2
     2107153.611      434084.961     2107503.067      434248.048
#Sta/Elev= 30
       0 2917.16     9.9 2913.16    19.8 2909.34    29.7 2905.76    39.6 2902.45
    49.4 2899.46    59.3 2896.67    69.2 2894.11    79.1 2891.82      89 2889.87
    98.9 2888.36   108.8 2887.28   128.6  2885.6   150.22884.316   168.1 2883.58
     178 2883.69   185.2 2884.97   187.9 2885.45   197.8 2889.66   207.6 2895.25
   237.3 2909.89   247.2 2914.25   257.1 2917.92     267 2921.07   276.9 2923.93
   296.6  2929.5   316.4 2934.86   336.2 2940.42   365.9 2949.28   385.6 2955.35
#Mann= 3 , 0 , 0
       0      .1       0   150.2    .045       0   185.2      .1       0
Bank Sta=150.2,185.2
XS Rating Curve= 0 ,0
Exp/Cntr=0.3,0.1

Type RM Length L Ch R = 1 ,14276.6 ,253.3,249.2,245.3
XS GIS Cut Line= 2
     2106981.781      434130.331     2107298.177      434551.353
#Sta/Elev= 30
       0 2953.75    59.6 2934.17    89.4 2924.58    99.4 2921.52   109.3 2918.74
   119.2 2916.15     149 2908.71     159 2905.83   168.9 2902.08   198.7 2889.48
   208.7 2885.86   219.42882.386   228.6 2879.93   238.5 2879.08   248.4    2880
   254.42882.058   258.4 2883.43   268.3 2888.18   278.2 2892.74   298.1 2900.06
     308 2903.57     318 2906.42   327.9 2908.45   377.6  2915.7   397.5 2918.87
   427.3  2924.1   457.1  2929.9     477 2934.02   496.8 2938.41   526.7 2945.28
#Mann= 3 , 0 , 0
       0      .1       0   219.4    .045       0   254.4      .1       0
Bank Sta=219.4,254.4
XS Rating Curve= 0 ,0
Exp/Cntr=0.3,0.1

Type RM Length L Ch R = 1 ,14027.4 ,372.2,373,360.5
XS GIS Cut Line= 2
      2106800.19      434337.235     2107117.498      434664.933
#Sta/Elev= 28
       0  2915.9    19.8 2911.58    49.6 2905.42    89.2 2897.67     119 2892.11
   128.9 2889.89   138.8 2887.27   158.7 2881.74   168.6 2879.22   178.5 2876.94
   188.4 2874.98   198.3 2873.35   210.6 2870.92   218.2  2869.4   228.1 2868.17
     238 2869.31   245.62872.588   247.9 2873.58   257.8  2878.8   267.7 2882.72
   287.6 2889.26   317.3 2899.32   327.2 2902.28     357 2909.43   396.6 2919.25
   416.5  2924.1   446.2  2931.3   456.2 2933.65
#Mann= 3 , 0 , 0
       0      .1       0   210.6    .045       0   245.6      .1       0
Bank Sta=210.6,245.6
XS Rating Curve= 0 ,0
Exp/Cntr=0.3,0.1

Type RM Length L Ch R = 1 ,13654.4 ,283.9,282.8,291
XS GIS Cut Line= 2
      2106491.21      434366.788     2106811.082      434805.916
#Sta/Elev= 30
       0 2951.76    20.1 2943.02    80.5 2917.33    90.6 2912.79   100.6 2907.61
   110.7  2901.8   120.7 2895.68   140.8 2883.09   150.9 2877.03     161  2871.4
     171 2866.38   181.1 2862.01   191.2 2858.17   201.2  2854.8   231.4 2845.96
   237.12844.605   241.5 2843.56   251.5 2842.82   261.6 2843.12   272.12844.414
   321.9  2851.8     332 2853.42   342.1 2855.32   352.1 2857.58   362.2 2860.34
   402.4 2873.09   412.5 2876.11   422.6 2878.76   432.6 2881.05   543.3 2904.95
#Mann= 3 , 0 , 0
       0      .1       0   237.1    .045       0   272.1      .1       0
Bank Sta=237.1,272.1
XS Rating Curve= 0 ,0
Exp/Cntr=0.3,0.1

Type RM Length L Ch R = 1 ,13371.6 ,273.2,278.7,285.8
XS GIS Cut Line= 2
     2106324.655      434628.705     2106691.036      435007.031
#Sta/Elev= 30
       0 2891.57     9.9 2887.94    29.8 2881.73    59.6 2871.79    69.6 2868.61
    89.4  2862.6   119.2 2854.12   129.2 2851.78   139.1 2849.68   228.6 2831.72
   245.8 2827.63   248.4 2827.05   258.4 2825.63   268.3 2825.83   278.2 2828.15
   280.82828.943   288.2  2831.2     308 2835.69     318 2838.66   327.9 2843.36
   337.8 2849.37   347.8 2855.68   367.7 2868.52   377.6 2873.73   387.5 2877.66
   437.2 2894.43   447.2 2897.45   457.1 2900.19   506.8 2912.44   526.7 2917.69
#Mann= 3 , 0 , 0
       0      .1       0   245.8    .045       0   280.8      .1       0
Bank Sta=245.8,280.8
XS Rating Curve= 0 ,0
Exp/Cntr=0.3,0.1

Type RM Length L Ch R = 1 ,13092.9 ,252.5,248.7,244.9
XS GIS Cut Line= 2
     2106175.712      434754.293     2106370.802      435165.347
#Sta/Elev= 30
       0  2873.6     9.9 2870.49    49.5 2859.99    98.9 2847.26   128.6 2839.45
   187.9 2824.12   197.8 2821.24   207.7 2817.62     210 2816.93   217.6 2814.65
   227.5 2813.92   237.4 2816.08     245 2819.98   247.3 2821.16   257.2 2827.16
   267.1 2832.96     277 2839.37   286.8 2846.14   296.7  2852.8   306.6 2859.04
   316.5 2864.22   326.4 2867.24   336.3 2868.98     366  2873.4   375.9 2875.04
   385.8  2877.3   395.6 2880.68   435.2 2896.82   445.1 2900.55     455  2903.9
#Mann= 3 , 0 , 0
       0      .1       0     210    .045       0     245      .1       0
Bank Sta=210,245
XS Rating Curve= 0 ,0
Exp/Cntr=0.3,0.1

Type RM Length L Ch R = 1 ,12844.3 ,257.9,247.5,237
XS GIS Cut Line= 2
     2105916.918      434874.027     2106177.696       435246.88
#Sta/Elev= 30
       0 2894.74    19.8 2885.56    29.7 2881.12    49.5 2872.56    69.2 2864.38
    79.1 2860.67    98.9 2854.09   108.8 2850.57   118.7  2846.8   128.6 2842.76
   138.5 2838.55   148.4 2834.24   168.2 2825.39   187.9 2816.34   197.8 2811.43
   207.7 2805.51     210 2804.59   217.6 2801.55   227.5 2800.56   237.4 2801.58
     245 2803.33     277 2811.39   286.8 2813.95   306.6 2819.33   326.4 2824.42
   405.5 2843.69   415.4  2846.4   425.3 2849.42   445.1 2855.96     455 2859.38
#Mann= 3 , 0 , 0
       0      .1       0     210    .045       0     245      .1       0
Bank Sta=210,245
XS Rating Curve= 0 ,0
Exp/Cntr=0.3,0.1

Type RM Length L Ch R = 1 ,12596.8 ,281,281.3,281.5
XS GIS Cut Line= 3
     2105689.759      435120.204     2105889.646      435228.839
     2106089.533      435337.474
#Sta/Elev= 27
       0 2866.59    29.7 2854.69    39.6 2850.52      89 2829.35   108.8 2820.58
   138.5 2807.19   148.4 2802.57   158.3 2797.42   168.2 2791.67   169.52791.146
     178 2787.72   187.9 2787.06   197.8 2788.54   204.52790.489   217.6 2794.35
   227.5 2796.71   267.1 2805.72   296.7  2812.6   306.6 2814.75   316.5 2816.61
   336.3 2820.08   385.8 2828.25   395.6 2829.97   405.5 2832.07   415.4 2834.82
   425.3 2838.16     455 2848.91
#Mann= 3 , 0 , 0
       0      .1       0   169.5    .045       0   204.5      .1       0
Bank Sta=169.5,204.5
XS Rating Curve= 0 ,0
Exp/Cntr=0.3,0.1

Type RM Length L Ch R = 1 ,12315.5 ,235.2,250.8,266.4
XS GIS Cut Line= 2
     2105555.612      435365.576     2105955.386      435582.845
#Sta/Elev= 29
       0 2813.28     9.9 2809.62    19.8 2806.12    29.7 2803.24    39.6 2800.87
    79.1 2791.93   118.7 2783.48   138.5 2779.64   158.3 2776.11   173.6 2773.17
     178 2772.33   187.9 2771.17   197.8 2771.56   207.7 2774.22   208.62774.588
   217.6 2778.27   227.5 2781.74   257.2 2790.03   286.8 2798.41   316.5 2806.41
   326.4 2808.99   336.3 2811.46   356.1 2816.24     366 2818.47   405.5 2826.74
   415.4 2829.06   425.3 2832.27   435.2  2836.3     455 2844.78
#Mann= 3 , 0 , 0
       0      .1       0   173.6    .045       0   208.6      .1       0
Bank Sta=173.6,208.6
XS Rating Curve= 0 ,0
Exp/Cntr=0.3,0.1

Type RM Length L Ch R = 1 ,12064.7 ,338.7,363,387.3
XS GIS Cut Line= 3
     2105471.443      435433.156     2105555.847      435644.419
     2105640.252      435855.682
#Sta/Elev= 30
       0 2806.73     9.9 2801.17    19.8 2796.12    29.7  2792.3    39.6 2789.87
    59.4 2786.12    69.2 2784.12   158.3 2765.57   168.2 2763.35   181.2 2759.75
   187.9 2757.99   197.8 2756.61   207.7 2756.86   216.22758.217   217.6 2758.44
   227.5  2760.8   237.4 2762.98     277 2770.34   296.7  2774.3   306.6 2776.12
   316.5 2777.39   326.4 2777.64   336.3 2777.19   346.2 2777.17   356.1  2777.8
     366  2779.8   385.8 2785.23   425.3 2796.67   435.2 2799.61     455 2805.73
#Mann= 3 , 0 , 0
       0      .1       0   181.2    .045       0   216.2      .1       0
Bank Sta=181.2,216.2
XS Rating Curve= 0 ,0
Exp/Cntr=0.3,0.1

Type RM Length L Ch R = 1 ,11701.7 ,115.3,124.9,135.5
XS GIS Cut Line= 3
     2105308.741      435534.113     2105155.998      435728.105
     2105184.154      435810.734
#Sta/Elev= 29
       0 2764.07    19.8  2761.1    29.6 2759.85    39.5 2758.84    59.3 2757.14
    69.1  2756.4      79 2755.68   108.6  2753.9   128.4 2752.31   138.3 2751.17
   148.1 2749.86   157.82748.322   167.9 2747.16   177.8 2746.75   192.82746.816
   197.5 2746.84   207.4 2747.36   217.3 2748.72   227.2 2750.33     237 2751.76
   246.9 2752.96   256.6 2754.69   266.3 2756.03     276  2756.8   285.7 2757.12
   305.1 2756.74   314.8 2756.73   324.5 2756.91   334.2 2757.28
#Mann= 3 , 0 , 0
       0      .1       0   157.8    .045       0   192.8      .1       0
Bank Sta=157.8,192.8
XS Rating Curve= 0 ,0
Exp/Cntr=0.3,0.1
